--- LostCrLR.prj (project) ---

Proj Title=LostCrLR
Current Plan=p01
Default Exp/Contr=0,0
English Units
Geom File=g01
Flow File=f01
Plan File=p01
BEGIN DESCRIPTION:
END DESCRIPTION:
DSS Export Rating Curves= 0
DSS Export Rating Curve Sorted= 0
DSS Export Volume Flow Curves= 0
DXF OffsetX= 0
DXF OffsetY= 0
DXF ScaleX= 0
DXF ScaleY= 0

--- LostCrLR.p01 (plan) ---

Plan Title=Floodplain
Program Version=4.00
Geom File=g01
Flow File=f01
K Sum by GR=0
Std Step Tol=0.01
Critical Tol=0.01
Num of Std Step Trials=20
Max Error Tol=0.3
Flow Tol Ratio=0.001
Split Flow NTrial=30
Split Flow Tol=0.02
Split Flow Ratio=0.02
Log Output Level=0
Friction Slope Method=1
Unsteady Friction Slope Method=2
Unsteady Bridges Friction Slope Method=1
Global Log Level=0
CheckData=False
Run HTab=0
Run UNet=0
Run PostProcess=0
UNET Theta=0
UNET Theta Warmup=0
UNET ZTol=0
UNET ZSATol=0
UNET MxIter=0
UNET MaxInSteps=0
UNET DtIC=0
UNET DtMin=0
UNET MaxCRTS=0
UNET WFStab=0
UNET SFStab=0
UNET WFX=0
UNET SFX=0
UNET DSS MLevel=0
UNET DZMax Abort=0
UNET Convert EG Bridges=0
UNET Use Existing IB Tables=0
UNET Froude Limit=0
UNET Froude Power=0
Write IC File=0
Echo Input=False
Echo Output=False
Write Detailed=0

--- LostCrLR.f01 (steady flow) ---

Flow Title=NFF Regression Equation
Program Version=4.00
Number of Profiles= 1
Profile Names=P100yr
River Rch & RM=LostCrLR,Main            ,27600.5
3244.379
River Rch & RM=LostCrLR,Main            ,24555.8
3524.856
River Rch & RM=LostCrLR,Main            ,18162.2
3752.042
River Rch & RM=LostCrLR,Main            ,12000.5
4168.797
River Rch & RM=LostCrLR,Main            ,8400.5
 4192.04
River Rch & RM=LostCrLR,Main            ,357.4
 4243.38
River Rch & RM=LostCrLR,Main            ,0.5
4245.936
Boundary for River Rch & Prof#=LostCrLR,Main            , 1
Up Type= 0
Dn Type= 3
Dn Slope=0.00277
DSS Import GetInterval= 0
DSS Import GetPeak= 0
DSS Import FillOption= 0

--- LostCrLR.g01 (geometry) ---

Geom Title=USGS 3m DEM
Program Version=4.00

River Reach=LostCrLR     ,Main
Reach XY= 30
     1724165.799      243443.649     1723448.579      244304.517
     1722325.811      244250.244     1721968.829      244529.420
     1721490.319      245725.231     1720835.144      246157.355
     1721043.354      246438.385     1720428.167      247611.570
     1720442.486      248894.191     1718051.741      251527.944
     1717960.335      250810.693     1717056.637      250476.840
     1716661.595      250809.747     1716288.921      250667.228
     1716250.297      250978.359     1715940.132      250889.483
     1715523.750      251237.763     1715056.636      250666.667
     1714459.799      251521.657     1714341.541      251132.600
     1713968.814      251284.511     1713824.629      252035.442
     1714362.223      252716.395     1713654.164      253135.501
     1713387.725      253610.528     1714590.243      253445.050
     1715527.406      254903.884     1716460.001      255163.241
     1716997.325      254620.939     1717402.136      255183.629

Type RM Length L Ch R = 1 ,27600.5,351.613,342.625,337.497
XS GIS Cut Line= 3
     1723919.859      243007.992     1724156.994      243448.390
     1724930.323      244363.662
#Sta/Elev= 30
       0 1164.90   133.1 1109.33   279.3 1051.97   329.8 1034.44   426.0 1010.21
   457.0 1001.55   467.9 1000.26   492.7  999.54   498.5  999.21   507.7  999.56
   572.3 1001.86   649.9 1000.93   908.8 1002.17   986.2 1001.71  1002.8 1002.39
  1116.1 1001.77  1168.0 1003.39  1215.2 1008.20  1267.9 1015.32  1293.9 1022.11
  1314.5 1024.70  1364.1 1040.65  1397.7 1050.06  1410.2 1052.39  1426.9 1053.15
  1488.3 1060.70  1536.2 1068.93  1554.7 1072.86  1610.5 1081.77  1698.4 1099.07
#Mann= 3 , 0 , 0
       0     0.1       0   492.7   0.045       0   507.7     0.1       0
Bank Sta=   492.7,   507.7
Exp/Cntr=0.3,0.1

Type RM Length L Ch R = 1 ,27257.8,555.302,569.811,584.988
XS GIS Cut Line= 3
     1723469.705      243141.355     1723892.515      243664.102
     1724907.261      244417.474
#Sta/Elev= 30
       0 1186.78    45.7 1178.34    68.4 1172.71    79.4 1171.12   121.8 1161.76
   225.8 1136.26   248.3 1129.64   265.1 1122.18   312.7 1095.02   332.7 1086.69
   388.6 1070.00   450.6 1049.66   586.5 1015.52   619.7 1006.05   653.5  997.88
   684.3  998.94   699.3  999.24   991.5 1004.25  1202.6 1005.43  1287.7 1004.68
  1345.5 1005.50  1376.8 1007.42  1434.1 1012.44  1494.1 1023.74  1518.7 1024.88
  1588.4 1038.77  1686.6 1054.01  1764.6 1063.37  1853.0 1080.22  1936.2 1098.43
#Mann= 3 , 0 , 0
       0     0.1       0   684.3   0.045       0   699.3     0.1       0
Bank Sta=   684.3,   699.3
Exp/Cntr=0.3,0.1

Type RM Length L Ch R = 1 ,26688,283.812,287.564,291.263
XS GIS Cut Line= 3
     1723464.291      243644.301     1723580.021      244084.154
     1723869.432      244984.340
#Sta/Elev= 30
       0 1064.73    48.4 1060.34   111.9 1056.75   211.0 1053.10   247.0 1049.52
   267.3 1045.03   276.3 1043.46   308.4 1035.98   382.0 1014.86   406.6 1008.50
   418.2 1006.54   442.9 1005.44   495.4  999.45   518.0  999.20   520.5  999.20
   535.5  999.24   608.9  999.72   742.5 1003.12   780.0 1011.68   804.9 1014.27
   917.7 1054.33  1009.9 1083.94  1039.0 1092.20  1046.3 1094.04  1187.6 1120.74
  1239.9 1133.24  1266.3 1138.59  1327.9 1152.48  1380.9 1166.45  1400.4 1170.32
#Mann= 3 , 0 , 0
       0     0.1       0   520.5   0.045       0   535.5     0.1       0
Bank Sta=   520.5,   535.5
Exp/Cntr=0.3,0.1

Type RM Length L Ch R = 1 ,26400.5,390.534,400,408.43
XS GIS Cut Line= 3
     1723321.841      243662.412     1723381.353      244327.017
     1723430.732      244814.104
#Sta/Elev= 30
       0 1058.84    90.5 1049.47   150.7 1045.29   185.8 1048.16   209.7 1046.65
   229.5 1043.57   262.6 1036.99   312.8 1025.98   343.2 1018.15   364.9 1014.11
   410.2 1006.89   445.9 1004.39   502.0 1001.57   528.1 1001.66   602.4 1003.57
   629.5 1003.44   650.8  999.74   659.8  999.44   670.8  999.36   674.8  999.45
   686.5  999.74   695.9 1001.73   717.4 1009.08   734.3 1015.39   758.7 1018.92
   799.6 1029.39   845.9 1043.31   955.3 1077.15  1027.4 1099.96  1156.8 1142.36
#Mann= 3 , 0 , 0
       0     0.1       0   659.8   0.045       0   674.8     0.1       0
Bank Sta=   659.8,   674.8
Exp/Cntr=0.3,0.1

Type RM Length L Ch R = 1 ,26000.5,335.85,330.064,325.579
XS GIS Cut Line= 3
     1723246.768      243541.103     1722992.848      244282.103
     1722855.799      244771.208
#Sta/Elev= 30
       0 1070.74   150.1 1051.15   244.3 1041.46   256.6 1041.11   310.3 1034.72
   453.3 1013.76   486.9 1010.36   543.9 1007.12   623.8 1004.09   666.2 1003.41
   724.0 1001.52   741.8 1002.04   751.2 1001.55   766.3 1000.09   775.8  999.70
   776.2  999.68   790.8 1002.13   828.8 1008.18   855.3 1011.24   924.8 1016.70
   944.7 1020.27   998.0 1028.05  1010.2 1030.68  1027.9 1035.48  1068.3 1048.93
  1084.1 1055.01  1120.9 1064.29  1146.8 1070.13  1219.8 1080.62  1291.2 1093.11
#Mann= 3 , 0 , 0
       0     0.1       0   775.8   0.045       0   790.8     0.1       0
Bank Sta=   775.8,   790.8
Exp/Cntr=0.3,0.1

Type RM Length L Ch R = 1 ,25670.4,611.161,594.891,576.95
XS GIS Cut Line= 3
     1722993.082      242449.483     1722669.932      244218.707
     1722624.084      244794.159
#Sta/Elev= 30
       0 1230.83    95.3 1205.17   153.9 1183.97   178.1 1179.05   223.0 1178.37
   242.9 1174.11   371.2 1128.07   519.8 1121.34   552.2 1115.57   629.5 1095.46
   703.8 1081.09   761.1 1072.12   833.6 1066.14  1039.8 1032.72  1106.4 1024.90
  1267.3 1022.76  1335.0 1015.19  1405.1 1001.26  1642.0 1003.45  1768.7 1000.67
  1813.7 1003.61  1828.7 1004.55  1864.3 1006.34  1890.7 1019.96  1902.4 1023.09
  2004.5 1028.90  2033.0 1033.68  2051.6 1032.07  2246.3 1069.61  2375.8 1083.76
#Mann= 3 , 0 , 0
       0     0.1       0  1813.7   0.045       0  1828.7     0.1       0
Bank Sta=  1813.7,  1828.7
Exp/Cntr=0.3,0.1

Type RM Length L Ch R = 1 ,25075.5,278.572,275.046,268.712
XS GIS Cut Line= 3
     1721332.589      243548.790     1722201.273      244432.849
     1722511.077      244816.273
#Sta/Elev= 30
       0 1271.74    38.1 1262.15    52.7 1256.87    96.7 1239.63   124.9 1226.22
   177.1 1203.45   244.0 1176.48   291.6 1159.99   368.9 1139.24   393.1 1134.21
   435.5 1131.26   471.9 1124.22   587.7 1095.52   701.8 1063.75   752.7 1048.47
   864.6 1012.18   896.6 1002.77   920.7  998.35  1218.5 1003.40  1233.5 1005.63
  1285.6 1019.17  1329.4 1024.98  1337.4 1025.93  1380.8 1025.16  1392.5 1026.55
  1422.5 1033.30  1513.5 1056.64  1580.5 1067.22  1620.0 1072.46  1732.4 1078.76
#Mann= 3 , 0 , 0
       0     0.1       0  1218.5   0.045       0  1233.5     0.1       0
Bank Sta=  1218.5,  1233.5
Exp/Cntr=0.3,0.1

Type RM Length L Ch R = 1 ,24800.5,246.573,244.611,244.298
XS GIS Cut Line= 3
     1721551.855      244263.980     1721954.731      244549.324
     1722385.772      244809.534
#Sta/Elev= 30
       0 1110.79    28.8 1102.57    83.4 1085.66   133.5 1070.62   213.6 1049.41
   239.5 1042.35   246.3 1040.92   382.5 1009.39   408.0 1003.78   431.9  998.92
   445.5  997.07   485.7  996.63   486.2  996.66   493.4  997.13   497.3  998.04
   501.2  999.32   526.7 1007.69   532.7 1010.14   562.7 1019.21   576.3 1021.43
   629.0 1023.49   662.5 1024.26   691.0 1024.65   733.7 1024.61   806.1 1028.95
   826.2 1031.90   872.7 1042.24   917.9 1051.97   973.0 1066.53   997.2 1071.24
#Mann= 3 , 0 , 0
       0     0.1       0   486.2   0.045       0   501.2     0.1       0
Bank Sta=   486.2,   501.2
Exp/Cntr=0.3,0.1

Type RM Length L Ch R = 1 ,24555.8,438.766,434.802,430.839
XS GIS Cut Line= 3
     1721384.450      244500.427     1721818.299      244750.016
     1722250.138      245003.021
#Sta/Elev= 30
       0 1143.24     7.7 1140.47    35.3 1128.92   125.9 1101.30   158.4 1091.00
   272.9 1055.91   312.1 1045.00   386.1 1026.12   442.3 1014.44   457.1 1011.12
   486.7 1005.68   527.6  998.78   536.2  998.28   548.6  997.64   551.2  998.03
   570.7 1000.98   608.2 1007.22   624.6 1009.08   654.3 1011.41   669.2 1012.21
   715.2 1013.10   751.7 1013.32   782.7 1016.01   873.2 1025.35   900.0 1026.51
   925.8 1025.20   933.6 1025.81   948.6 1027.24   969.4 1031.53  1001.0 1039.76
#Mann= 3 , 0 , 0
       0     0.1       0   536.2   0.045       0   551.2     0.1       0
Bank Sta=   536.2,   551.2
Exp/Cntr=0.3,0.1

Type RM Length L Ch R = 1 ,24121,516.164,520.587,521.211
XS GIS Cut Line= 3
     1721222.178      244997.264     1721691.534      245170.918
     1722155.708      245358.863
#Sta/Elev= 30
       0 1111.31   160.7 1071.77   266.6 1049.78   294.1 1045.26   327.0 1042.52
   344.7 1040.36   374.5 1033.30   410.2 1020.34   426.1 1011.18   447.2 1001.59
   457.4  999.18   472.4  999.25   476.5  999.25   504.4 1001.50   638.3 1008.94
   664.2 1011.53   721.4 1013.71   767.0 1017.38   818.2 1024.37   846.3 1028.90
   868.0 1031.95   883.9 1033.04   901.6 1033.78   922.7 1039.00   934.4 1043.47
   949.3 1047.16   957.7 1049.66   965.1 1050.18   991.9 1054.80  1001.2 1055.20
#Mann= 3 , 0 , 0
       0     0.1       0   457.4   0.045       0   472.4     0.1       0
Bank Sta=   457.4,   472.4
Exp/Cntr=0.3,0.1

Type RM Length L Ch R = 1 ,23600.5,396.456,400,408.691
XS GIS Cut Line= 3
     1721056.976      245381.379     1721514.796      245656.729
     1722009.086      245855.030
#Sta/Elev= 30
       0 1066.92    26.1 1063.49    60.2 1056.74    71.3 1054.05    79.1 1051.55
   120.7 1044.54   189.9 1031.81   228.4 1015.85   241.8 1013.38   389.9 1010.01
   467.4 1007.57   504.0 1007.13   526.7 1004.53   533.1 1003.87   541.7 1004.21
   576.2 1010.61   582.6 1011.51   614.0 1014.17   744.0 1021.57   776.1 1024.47
   800.8 1025.96   840.9 1031.59   852.4 1032.81   861.5 1033.74   899.9 1036.31
   934.9 1040.80  1008.5 1051.62  1011.9 1052.37  1040.6 1054.81  1066.8 1058.99
#Mann= 3 , 0 , 0
       0     0.1       0   526.7   0.045       0   541.7     0.1       0
Bank Sta=   526.7,   541.7
Exp/Cntr=0.3,0.1

Type RM Length L Ch R = 1 ,23200.5,344.098,336.897,328.349
XS GIS Cut Line= 3
     1720802.154      245524.469     1721216.381      245894.035
     1721600.418      246274.053
#Sta/Elev= 30
       0 1082.37    34.1 1072.65    87.6 1059.55   156.5 1050.28   210.4 1037.97
   228.6 1030.94   252.1 1021.43   284.4 1015.64   296.5 1014.71   415.6 1010.73
   461.4 1009.61   526.4 1008.34   547.6 1005.95   554.1 1005.19   562.6 1005.30
   566.4 1005.35   617.2 1009.79   643.7 1013.47   661.5 1018.81   722.2 1035.74
   740.0 1039.30   785.2 1046.75   797.8 1048.59   811.5 1049.92   846.6 1049.20
   935.7 1040.23   960.2 1040.07   981.7 1041.84  1041.2 1047.48  1095.4 1051.85
#Mann= 3 , 0 , 0
       0     0.1       0   547.6   0.045       0   562.6     0.1       0
Bank Sta=   547.6,   562.6
Exp/Cntr=0.3,0.1

Type RM Length L Ch R = 1 ,22863.6,635.849,637.911,640.956
XS GIS Cut Line= 3
     1720513.254      245801.235     1720879.356      246035.360
     1721525.152      246342.076
#Sta/Elev= 30
       0 1056.32    50.0 1051.93    71.1 1049.44   104.7 1047.27   121.1 1047.02
   182.5 1044.23   190.7 1043.36   201.3 1043.11   215.3 1042.04   247.8 1035.51
   281.0 1025.02   302.0 1019.02   319.6 1014.64   358.1 1011.29   473.5 1005.76
   484.6 1005.22   488.5 1005.27   652.0 1007.47   706.1 1009.56   751.4 1010.73
   757.6 1012.07   825.2 1021.27   848.3 1020.60   881.8 1021.26   949.9 1024.60
   967.1 1024.10  1008.2 1026.53  1063.5 1033.43  1112.4 1041.51  1149.5 1046.53
#Mann= 3 , 0 , 0
       0     0.1       0   473.5   0.045       0   488.5     0.1       0
Bank Sta=   473.5,   488.5
Exp/Cntr=0.3,0.1

Type RM Length L Ch R = 1 ,22225.6,227.941,225.192,226.606
XS GIS Cut Line= 3
     1720210.220      246239.403     1720963.591      246531.527
     1721455.589      246815.963
#Sta/Elev= 30
       0 1072.45    45.4 1072.62    82.2 1069.06   125.7 1062.33   156.3 1059.36
   229.4 1057.88   290.1 1053.82   304.2 1051.42   324.3 1050.61   343.8 1047.71
   375.2 1040.40   447.4 1011.85   462.9 1008.07   548.3 1006.39   687.9 1007.10
   817.1 1002.60   832.1 1002.22   833.6 1002.18   845.4 1003.45   868.4 1014.43
   880.7 1018.23   904.2 1019.25   917.9 1022.59   946.6 1038.03   964.0 1045.58
   991.9 1052.23  1151.4 1059.77  1273.2 1064.25  1311.6 1065.00  1376.3 1062.73
#Mann= 3 , 0 , 0
       0     0.1       0   817.1   0.045       0   832.1     0.1       0
Bank Sta=   817.1,   832.1
Exp/Cntr=0.3,0.1

Type RM Length L Ch R = 1 ,22000.5,398.984,400,393.279
XS GIS Cut Line= 3
     1720373.112      246535.921     1720840.280      246713.492
     1721269.224      246998.954
#Sta/Elev= 30
       0 1073.35    16.6 1070.98    84.0 1058.51   103.1 1054.52   121.8 1047.36
   136.3 1042.44   149.2 1036.21   179.5 1022.93   211.1 1010.47   213.4 1009.59
   225.4 1007.36   348.7 1005.69   420.5 1005.47   479.4 1002.97   492.3 1003.06
   507.3 1002.96   547.2 1002.74   562.5 1003.98   585.5 1008.32   600.8 1016.20
   626.3 1031.36   641.4 1039.73   646.4 1042.22   665.8 1049.10   680.8 1050.14
   705.1 1052.47   769.8 1056.50   854.6 1060.23   910.8 1061.78  1015.0 1060.70
#Mann= 3 , 0 , 0
       0     0.1       0   492.3   0.045       0   507.3     0.1       0
Bank Sta=   492.3,   507.3
Exp/Cntr=0.3,0.1

Type RM Length L Ch R = 1 ,21600.5,404.787,400,404.375
XS GIS Cut Line= 3
     1720236.099      246888.908     1720695.519      247085.571
     1721179.227      247229.895
#Sta/Elev= 30
       0 1064.48    16.6 1060.88    44.7 1056.71    90.1 1043.49   145.0 1023.61
   182.0 1010.87   188.3 1009.50   263.5 1006.69   377.6 1005.50   477.3 1005.76
   492.2 1002.99   498.5 1002.27   507.2 1002.56   544.2 1004.44   550.2 1006.49
   556.6 1006.99   562.1 1008.73   593.8 1027.96   607.6 1033.59   642.6 1038.45
   666.2 1039.65   744.7 1040.32   770.3 1043.70   787.9 1044.06   815.4 1041.23
   884.7 1038.14   921.4 1033.77   971.2 1029.61   994.6 1026.50  1004.5 1026.32
#Mann= 3 , 0 , 0
       0     0.1       0   492.2   0.045       0   507.2     0.1       0
Bank Sta=   492.2,   507.2
Exp/Cntr=0.3,0.1

Type RM Length L Ch R = 1 ,21200.5,409.457,400,387.594
XS GIS Cut Line= 3
     1720017.083      247301.394     1720503.662      247399.728
     1720981.107      247636.374
#Sta/Elev= 30
       0 1051.34    36.2 1044.53    62.2 1041.01    82.6 1037.07    93.7 1035.62
   163.0 1025.01   219.3 1012.50   232.3 1009.36   245.1 1006.96   346.6 1002.84
   458.1 1000.34   488.9 1001.84   503.9 1002.48   572.6 1002.34   604.9 1003.88
   612.3 1003.97   616.5 1004.66   634.6 1009.49   643.1 1012.30   676.2 1021.75
   678.6 1022.21   735.7 1029.39   773.4 1032.56   834.4 1031.98   864.6 1032.30
   906.6 1033.80   923.4 1035.11   977.2 1037.64  1010.3 1037.61  1029.3 1036.27
#Mann= 3 , 0 , 0
       0     0.1       0   488.9   0.045       0   503.9     0.1       0
Bank Sta=   488.9,   503.9
Exp/Cntr=0.3,0.1

Type RM Length L Ch R = 1 ,20800.5,400.562,400,393.257
XS GIS Cut Line= 3
     1719958.983      247884.129     1720444.779      247776.672
     1720961.551      247746.855
#Sta/Elev= 30
       0 1046.28     3.7 1045.34    66.2 1036.91   120.7 1031.25   157.0 1025.38
   183.2 1023.60   202.2 1024.02   264.0 1020.58   307.9 1018.58   311.6 1018.11
   331.5 1011.29   348.1 1004.92   381.2 1000.13   396.1 1000.67   444.7 1003.46
   473.2 1002.90     490 1001.63     505 1000.46   567.0 1001.83   595.3 1002.84
   601.1 1003.63   608.2 1005.39   655.9 1020.88   671.3 1025.06   678.0 1026.65
   721.3 1032.68   793.9 1036.93   904.2 1041.26   988.9 1040.27  1015.2 1039.07
#Mann= 3 , 0 , 0
       0     0.1       0     490   0.045       0     505     0.1       0
Bank Sta=     490,     505
Exp/Cntr=0.3,0.1

Type RM Length L Ch R = 1 ,20400.5,519.637,531.136,545.192
XS GIS Cut Line= 3
     1719848.669      248331.114     1720567.031      248152.572
     1721032.844      247979.638
#Sta/Elev= 30
       0 1081.21    24.3 1073.06    78.8 1057.37   155.0 1031.86   179.1 1022.90
   235.0 1003.84   251.4 1002.43   305.7 1003.80   360.3 1003.64   381.4 1002.52
   416.4 1004.57   497.1 1006.03   603.7 1000.41   630.0  999.78   708.5 1002.70
   732.7 1001.08   747.7 1000.07   759.2 1001.22   768.0 1005.65   783.4 1016.96
   788.3 1019.49   801.2 1024.39   814.2 1025.86   907.1 1026.95   962.7 1029.26
  1014.9 1030.16  1069.9 1028.05  1100.0 1029.29  1163.4 1035.62  1237.1 1045.92
#Mann= 3 , 0 , 0
       0     0.1       0   732.7   0.045       0   747.7     0.1       0
Bank Sta=   732.7,   747.7
Exp/Cntr=0.3,0.1

Type RM Length L Ch R = 1 ,19869.3,259.411,266.55,273.688
XS GIS Cut Line= 3
     1719900.559      248508.406     1720555.889      248686.347
     1721262.682      248841.370
#Sta/Elev= 30
       0 1082.32     8.6 1078.91    70.4 1064.38   125.4 1047.58   145.2 1040.23
   173.9 1031.73   203.6 1019.12   235.7 1004.05   247.3 1001.78   353.9 1002.96
   462.8 1002.56   566.4 1000.30   574.9 1000.09   581.4 1000.57   747.7 1003.15
   812.0 1005.76   821.6 1007.20   829.2 1008.42   858.4 1021.70   877.8 1028.86
   890.6 1031.09   921.7 1033.11   954.5 1037.73  1078.1 1058.69  1096.6 1060.90
  1133.0 1061.77  1138.2 1062.83  1263.1 1089.35  1324.3 1108.54  1402.7 1127.85
#Mann= 3 , 0 , 0
       0     0.1       0   566.4   0.045       0   581.4     0.1       0
Bank Sta=   566.4,   581.4
Exp/Cntr=0.3,0.1

Type RM Length L Ch R = 1 ,19602.8,398.298,402.314,405.829
XS GIS Cut Line= 3
     1719809.751      248521.379     1720686.842      249083.765
     1721094.278      249152.952
#Sta/Elev= 30
       0 1115.26    45.1 1103.24   100.9 1082.86   186.1 1058.61   218.2 1045.89
   259.2 1037.42   293.3 1027.15   341.2 1008.41   355.3 1005.15   405.8 1001.62
   469.4 1002.55   690.8 1002.49   722.2 1000.35   730.4  999.28   737.2 1000.32
   756.8 1003.11   923.3 1006.18   941.3 1008.98   970.9 1018.77   980.7 1020.61
  1032.3 1022.87  1084.1 1029.73  1175.9 1030.49  1226.3 1032.77  1259.1 1032.02
  1286.6 1027.80  1302.2 1027.49  1312.5 1028.09  1345.8 1033.51  1455.1 1039.49
#Mann= 3 , 0 , 0
       0     0.1       0   722.2   0.045       0   737.2     0.1       0
Bank Sta=   722.2,   737.2
Exp/Cntr=0.3,0.1

Type RM Length L Ch R = 1 ,19200.5,381.596,400,400.985
XS GIS Cut Line= 4
     1719462.688      248530.459     1719731.203      248781.951
     1720084.641      249112.981     1720848.279      249798.699
#Sta/Elev= 30
       0 1170.21     9.4 1170.73    44.8 1167.55   153.3 1150.75   181.0 1144.90
   283.5 1117.77   350.3 1091.83   396.4 1075.52   452.0 1061.48   518.3 1048.41
   571.2 1035.78   632.3 1025.43   667.1 1023.74   673.9 1022.28   723.0 1003.78
   745.6 1000.49   844.6 1000.17   859.6  999.86   931.5  998.10   987.0  998.18
  1075.4 1002.00  1130.7  998.37  1167.5 1002.20  1228.6 1006.16  1279.4 1020.66
  1495.7 1037.11  1614.3 1049.92  1752.3 1076.26  1822.7 1085.41  1878.5 1097.06
#Mann= 3 , 0 , 0
       0     0.1       0   844.6   0.045       0   859.6     0.1       0
Bank Sta=   844.6,   859.6
Exp/Cntr=0.3,0.1

Type RM Length L Ch R = 1 ,18800.5,647.927,638.247,646.488
XS GIS Cut Line= 3
     1719123.548      248373.539     1720049.595      249477.186
     1720931.509      250190.192
#Sta/Elev= 30
       0 1190.56    55.3 1185.17    92.2 1166.86   105.2 1164.44   124.6 1166.23
   141.4 1172.62   158.3 1175.46   259.6 1171.94   444.8 1146.80   694.2 1067.86
   891.4 1034.29   974.8 1028.61  1190.7 1027.02  1255.9 1021.10  1274.3 1016.78
  1312.1 1002.08  1433.2  998.82  1448.2  998.55  1543.7  996.61  1556.6  998.60
  1593.3 1014.39  1616.5 1021.88  1716.5 1023.77  1879.8 1036.39  2005.5 1040.58
  2111.6 1078.55  2211.6 1101.52  2410.1 1136.66  2465.5 1143.53  2574.8 1148.51
#Mann= 3 , 0 , 0
       0     0.1       0  1433.2   0.045       0  1448.2     0.1       0
Bank Sta=  1433.2,  1448.2
Exp/Cntr=0.3,0.1

Type RM Length L Ch R = 1 ,18162.2,482.677,476.536,470.394
XS GIS Cut Line= 2
     1719036.627      248616.919     1720192.679      251146.325
#Sta/Elev= 30
       0 1137.25    26.0 1136.83    40.3 1133.30    76.6 1121.79   130.8 1108.63
   153.5 1093.88   176.7 1090.48   274.2 1067.56   330.1 1061.30   386.3 1050.62
   438.5 1046.19   464.5 1041.96   625.2 1031.13   847.0 1023.51  1248.2 1021.29
  1347.7 1018.06  1421.4  997.34  1436.4  996.78  1438.4  996.70  1484.9 1000.02
  1560.9  999.54  1600.5 1004.15  1628.8 1002.58  1690.4 1006.55  1924.6 1013.66
  2028.7 1014.20  2378.0 1026.07  2512.0 1033.97  2709.6 1064.11  2781.1 1080.61
#Mann= 3 , 0 , 0
       0     0.1       0  1421.4   0.045       0  1436.4     0.1       0
Bank Sta=  1421.4,  1436.4
Exp/Cntr=0.3,0.1

Type RM Length L Ch R = 1 ,17685.7,488.195,485.217,483.768
XS GIS Cut Line= 2
     1718411.403      249166.404     1720115.105      251195.813
#Sta/Elev= 30
       0 1208.12    27.2 1206.40   126.3 1205.79   276.5 1181.69   387.5 1148.80
   446.0 1129.03   516.5 1101.48   620.2 1074.30   678.2 1056.87   753.0 1040.44
   857.1 1031.20   974.1 1017.49  1010.9 1015.89  1069.2 1016.65  1158.0 1010.64
  1217.4 1012.75  1239.2 1009.51  1294.3  996.67  1298.6  995.53  1309.3  995.88
  1354.9 1004.73  1427.8 1007.16  1463.0 1011.22  2025.5 1021.43  2268.8 1032.19
  2302.5 1035.68  2438.5 1056.38  2517.9 1072.30  2562.5 1084.33  2649.7 1103.21
#Mann= 3 , 0 , 0
       0     0.1       0  1294.3   0.045       0  1309.3     0.1       0
Bank Sta=  1294.3,  1309.3
Exp/Cntr=0.3,0.1

Type RM Length L Ch R = 1 ,17200.5,346.876,350.724,350.442
XS GIS Cut Line= 4
     1718393.411      250016.349     1718877.693      250460.451
     1719241.594      250842.002     1719787.403      251414.285
#Sta/Elev= 30
       0 1179.77   174.9 1147.56   225.7 1141.41   289.4 1118.22   353.1 1097.71
   380.2 1085.72   414.0 1065.74   443.8 1050.42   458.4 1044.91   502.5 1029.90
   575.1 1010.29   594.6 1006.96   630.8  997.71   649.6  994.78   655.5  993.90
   664.6  995.15   719.3 1002.02   788.8 1005.75  1003.1 1009.27  1191.9 1015.10
  1303.1 1020.31  1494.3 1033.48  1634.8 1052.60  1718.5 1072.23  1747.6 1077.65
  1821.4 1084.20  1855.0 1090.29  1871.7 1093.70  1922.0 1113.78  1975.2 1130.36
#Mann= 3 , 0 , 0
       0     0.1       0   649.6   0.045       0   664.6     0.1       0
Bank Sta=   649.6,   664.6
Exp/Cntr=0.3,0.1

Type RM Length L Ch R = 1 ,16849.7,389.566,400.465,413.87
XS GIS Cut Line= 4
     1718354.610      250312.784     1718715.019      250763.871
     1719060.139      251107.345     1719607.390      251552.643
#Sta/Elev= 30
       0 1171.61    45.1 1165.73    57.5 1163.63   138.0 1144.53   149.1 1141.21
   166.5 1137.17   183.6 1131.29   237.0 1109.41   270.2 1099.82   297.4 1090.09
   346.2 1067.14   427.1 1031.06   464.5 1018.12   511.9 1002.69   557.1  994.87
   567.7  994.61   582.7  994.34   584.3  994.31   611.3  999.48  1126.1 1013.76
  1241.3 1017.79  1286.6 1024.69  1344.6 1032.03  1381.1 1037.82  1413.2 1045.95
  1513.9 1075.15  1596.7 1096.10  1636.2 1106.73  1724.1 1125.14  1769.8 1131.08
#Mann= 3 , 0 , 0
       0     0.1       0   567.7   0.045       0   582.7     0.1       0
Bank Sta=   567.7,   582.7
Exp/Cntr=0.3,0.1

Type RM Length L Ch R = 1 ,16449.3,324.035,326.463,319.21
XS GIS Cut Line= 3
     1718285.810      250377.908     1718588.164      251428.442
     1719132.241      252241.531
#Sta/Elev= 30
       0 1150.47    61.4 1142.10    95.9 1129.72   196.8 1091.31   209.6 1086.95
   234.8 1082.67   256.7 1076.23   302.1 1058.07   308.4 1056.07   363.9 1040.85
   407.3 1030.25   555.5 1000.93   657.3  999.33   691.4  996.48     737  993.84
   737.6  993.81     752  994.09   782.0 1001.17   801.0 1002.53   945.4 1003.57
  1041.8 1005.77  1075.5 1007.48  1246.9 1012.35  1337.9 1018.67  1561.4 1028.21
  1615.3 1033.46  1713.3 1041.42  1770.0 1048.67  1869.8 1064.61  2071.5 1103.85
#Mann= 3 , 0 , 0
       0     0.1       0     737   0.045       0     752     0.1       0
Bank Sta=     737,     752
Exp/Cntr=0.3,0.1

Type RM Length L Ch R = 1 ,16122.8,1220.366,1232.064,1253.54
XS GIS Cut Line= 4
     1718214.152      250421.595     1718176.108      250902.945
     1718254.337      251311.475     1718906.246      252467.526
#Sta/Elev= 30
       0 1130.38    16.0 1124.86    63.0 1103.04   111.9 1076.68   122.5 1070.25
   148.9 1057.32   177.5 1048.89   223.3 1037.18   290.5 1022.97   398.4 1004.89
   420.4 1003.57   574.7 1000.04   833.2 1000.80   876.6  994.92   892.2  993.95
   892.6  993.92   907.2  994.39   918.3  994.79   956.0  999.40  1003.1 1001.28
  1320.0 1006.90  1467.7 1014.14  1603.5 1023.67  1670.8 1030.86  1707.5 1033.45
  1851.1 1049.78  2003.9 1065.99  2027.8 1069.32  2200.6 1098.53  2226.0 1104.02
#Mann= 3 , 0 , 0
       0     0.1       0   892.2   0.045       0   907.2     0.1       0
Bank Sta=   892.2,   907.2
Exp/Cntr=0.3,0.1

Type RM Length L Ch R = 1 ,14890.7,473.69,468.03,460.26
XS GIS Cut Line= 3
     1718223.128      250290.743     1717983.139      250711.758
     1717248.366      252324.784
#Sta/Elev= 30
       0 1158.98    56.4 1147.53    83.9 1140.15   113.5 1130.41   148.6 1117.82
   213.0 1084.91   240.5 1076.88   276.4 1061.18   345.9 1038.25   507.4 1001.05
   570.5  990.97   574.1  991.02   589.1  991.25   636.2  996.92   715.6 1003.45
  1041.2 1012.97  1119.0 1014.08  1202.0 1019.34  1332.5 1023.27  1398.8 1027.70
  1446.5 1028.21  1486.3 1032.19  1512.9 1037.84  1527.8 1038.32  1599.4 1045.19
  1702.6 1046.73  1783.2 1051.29  1999.6 1052.59  2149.0 1066.60  2257.1 1080.21
#Mann= 3 , 0 , 0
       0     0.1       0   574.1   0.045       0   589.1     0.1       0
Bank Sta=   574.1,   589.1
Exp/Cntr=0.3,0.1

Type RM Length L Ch R = 1 ,14422.7,529.674,526.787,526.01
XS GIS Cut Line= 3
     1717667.597      250021.930     1717551.906      250541.055
     1717465.013      251584.042
#Sta/Elev= 30
       0 1179.56    32.6 1173.51    83.0 1161.93   141.9 1150.89   191.7 1138.55
   228.5 1127.73   251.9 1119.27   282.2 1103.81   345.1 1067.46   387.3 1045.24
   431.4 1031.07   446.1 1024.26   475.8 1007.79   490.1 1001.42   507.0  996.37
   531.6  990.98   543.2  990.60   546.6  990.88   619.3  999.58   650.4 1001.93
   741.1 1003.83  1043.6 1007.02  1103.1 1006.83  1226.1 1013.45  1345.3 1016.55
  1387.5 1023.01  1414.8 1024.59  1448.6 1030.13  1484.4 1033.14  1578.5 1035.67
#Mann= 3 , 0 , 0
       0     0.1       0   531.6   0.045       0   546.6     0.1       0
Bank Sta=   531.6,   546.6
Exp/Cntr=0.3,0.1

Type RM Length L Ch R = 1 ,13895.9,704.788,695.467,687.206
XS GIS Cut Line= 3
     1717135.554      249949.572     1717033.469      250425.798
     1716980.964      251503.051
#Sta/Elev= 30
       0 1105.31    25.5 1106.32    59.8 1098.71   104.6 1086.24   185.6 1059.58
   215.5 1049.09   231.7 1041.12   243.0 1034.32   259.5 1028.89   275.5 1026.97
   295.5 1025.97   322.3 1021.87   336.0 1018.05   358.8 1014.50   418.3 1007.62
   456.0 1000.45   524.5  991.18   530.5  990.95   542.2  990.52   545.5  990.52
   777.6  994.53   939.2  999.74   988.8 1005.67  1107.1 1005.66  1206.9 1007.60
  1338.8 1008.72  1368.6 1010.23  1429.9 1014.93  1455.5 1016.26  1565.6 1020.07
#Mann= 3 , 0 , 0
       0     0.1       0   530.5   0.045       0   545.5     0.1       0
Bank Sta=   530.5,   545.5
Exp/Cntr=0.3,0.1

Type RM Length L Ch R = 1 ,13200.5,398.1,400,395.906
XS GIS Cut Line= 3
     1716289.918      250103.271     1716537.513      250818.702
     1716794.061      251667.852
#Sta/Elev= 30
       0 1082.77    60.6 1082.32    75.5 1081.30   101.1 1076.60   172.0 1060.84
   190.1 1056.68   241.4 1043.68   249.6 1040.99   300.1 1021.46   329.2 1009.24
   346.2 1003.18   349.6 1002.60   361.7 1001.27   449.8  997.86   487.8  997.10
   559.2  997.99   663.0  992.07   749.6  988.60   751.6  988.50   764.6  989.10
   776.5  989.75   819.4  996.36   838.5  999.51   877.1 1007.30   917.2 1014.06
   941.2 1014.43  1061.8 1013.24  1132.2 1011.09  1435.8 1016.36  1644.1 1022.08
#Mann= 3 , 0 , 0
       0     0.1       0   749.6   0.045       0   764.6     0.1       0
Bank Sta=   749.6,   764.6
Exp/Cntr=0.3,0.1

Type RM Length L Ch R = 1 ,12800.5,798.358,800,807.026
XS GIS Cut Line= 3
     1716063.923      250181.500     1716225.766      250718.605
     1716759.293      251746.081
#Sta/Elev= 30
       0 1100.93     7.1 1100.59    93.4 1084.13   139.8 1074.45   188.7 1062.44
   242.2 1051.92   291.9 1040.78   301.8 1037.78   330.7 1030.62   440.7  999.89
   494.6  996.71   526.7  995.32   553.5  990.24   559.5  988.99   568.5  990.29
   586.0  992.82   591.8  992.86   636.0  992.56   706.6  991.29   745.0  989.54
   801.7  991.61   832.8  993.31   857.5  996.15   957.1 1012.05   989.5 1014.30
  1206.4 1013.11  1439.1 1016.92  1502.7 1016.86  1587.6 1019.68  1718.7 1023.26
#Mann= 3 , 0 , 0
       0     0.1       0   553.5   0.045       0   568.5     0.1       0
Bank Sta=   553.5,   568.5
Exp/Cntr=0.3,0.1

Type RM Length L Ch R = 1 ,12000.5,270.204,273.099,275.1
XS GIS Cut Line= 3
     1715594.549      250016.349     1715844.903      250970.152
     1716063.923      251902.539
#Sta/Elev= 30
       0 1106.78    62.2 1087.64   141.8 1071.27   296.4 1036.28   333.2 1029.18
   439.1 1012.45   651.6 1004.35   676.9 1005.96   698.0 1006.14   925.2 1000.29
   944.7  999.10   954.4  996.50   967.4  990.19   978.6  988.62   993.6  988.35
   998.1  988.31  1044.2  991.35  1109.9  991.08  1173.3  994.32  1330.5  998.77
  1431.1 1013.41  1459.4 1016.69  1494.3 1024.08  1516.8 1029.99  1570.5 1033.94
  1715.6 1032.81  1727.7 1033.98  1752.1 1040.38  1792.4 1039.75  1943.9 1048.68
#Mann= 3 , 0 , 0
       0     0.1       0   978.6   0.045       0   993.6     0.1       0
Bank Sta=   978.6,   993.6
Exp/Cntr=0.3,0.1

Type RM Length L Ch R = 1 ,11727.4,977.698,970.476,963.305
XS GIS Cut Line= 3
     1715333.785      250190.192     1715638.010      251102.864
     1715777.084      251893.847
#Sta/Elev= 30
       0 1075.05    61.1 1058.80    73.0 1056.16   103.8 1046.89   134.7 1038.56
   306.0 1005.24   481.9  998.79   614.6  999.92   782.2  998.34   870.6  993.20
   894.9  992.17   971.0  990.81   992.7  988.51  1002.1  988.38    1008  988.66
    1023  989.05  1102.3  989.48  1140.9  991.86  1224.4  994.73  1283.0  994.45
  1304.0  994.70  1319.3  995.67  1347.2 1002.31  1420.5 1029.32  1454.0 1034.98
  1528.6 1044.71  1572.4 1048.85  1590.0 1052.94  1619.4 1056.88  1765.2 1071.85
#Mann= 3 , 0 , 0
       0     0.1       0    1008   0.045       0    1023     0.1       0
Bank Sta=    1008,    1023
Exp/Cntr=0.3,0.1

Type RM Length L Ch R = 1 ,10756.9,359.427,356.425,355.089
XS GIS Cut Line= 4
     1714542.803      250025.041     1715020.869      250668.258
     1715255.556      251320.167     1715620.625      252050.305
#Sta/Elev= 30
       0 1256.44    23.2 1256.93    34.1 1254.48    93.1 1231.78   142.1 1222.11
   285.7 1181.60   480.0 1138.92   545.5 1119.30   600.1 1100.25   664.2 1071.15
   679.0 1062.78   728.4 1022.53   755.4 1004.40   773.4  995.77   790.2  990.99
   817.6  988.84   832.6  988.41   834.6  988.39   864.6  994.64  1075.8 1007.06
  1358.3 1028.71  1478.8 1031.81  1573.0 1037.66  1673.1 1047.15  1898.6 1046.84
  1986.4 1057.11  2025.7 1059.16  2109.3 1071.44  2264.3 1082.85  2310.6 1088.63
#Mann= 3 , 0 , 0
       0     0.1       0   817.6   0.045       0   832.6     0.1       0
Bank Sta=   817.6,   832.6
Exp/Cntr=0.3,0.1

Type RM Length L Ch R = 1 ,10400.5,402.166,400,392.829
XS GIS Cut Line= 3
     1714568.879      250503.108     1714843.886      250994.147
     1715246.864      251824.310
#Sta/Elev= 30
       0 1174.74    13.0 1169.59   144.0 1134.41   170.5 1124.03   228.9 1104.45
   243.6 1099.14   342.2 1057.44   350.0 1054.92   369.4 1047.53   382.7 1043.48
   519.6  995.44   544.3  989.61   555.3  988.51   562.8  987.77   570.3  988.60
   580.8  989.32   612.5  993.74   654.2  996.51   701.3  998.66   884.4 1009.30
   936.1 1014.93   970.3 1019.41  1020.1 1027.47  1098.2 1041.34  1127.5 1043.71
  1253.8 1046.90  1299.4 1047.66  1318.3 1047.45  1349.9 1049.51  1485.6 1054.53
#Mann= 3 , 0 , 0
       0     0.1       0   555.3   0.045       0   570.3     0.1       0
Bank Sta=   555.3,   570.3
Exp/Cntr=0.3,0.1

Type RM Length L Ch R = 1 ,10000.5,1612.483,1600,1586.763
XS GIS Cut Line= 3
     1714221.195      250703.027     1714632.313      251330.963
     1715264.249      252067.689
#Sta/Elev= 30
       0 1181.77    36.6 1174.53    61.2 1167.33    77.2 1159.13    99.5 1140.45
   129.6 1110.41   177.1 1074.89   216.2 1050.56   226.2 1045.49   298.0 1017.76
   338.4 1005.74   373.4  997.47   387.6  996.22   519.2  993.55   569.5  995.25
   698.6  993.31   714.8  992.27     743  986.84   750.5  985.88     758  986.79
   824.6  992.88   914.6  997.53  1047.4 1022.54  1100.9 1031.00  1320.2 1044.49
  1365.3 1044.16  1576.3 1049.74  1658.0 1050.68  1699.9 1051.87  1721.2 1054.37
#Mann= 3 , 0 , 0
       0     0.1       0     743   0.045       0     758     0.1       0
Bank Sta=     743,     758
Exp/Cntr=0.3,0.1

Type RM Length L Ch R = 1 ,8400.5,641.817,630.544,622.735
XS GIS Cut Line= 3
     1713488.484      251474.215     1713881.781      251682.258
     1715272.941      252171.994
#Sta/Elev= 30
       0 1114.39    68.0 1088.57   141.5 1056.31   153.1 1052.27   347.3  998.09
   398.9  985.79   415.3  982.77   420.1  981.90   437.4  981.72   452.4  981.57
   453.5  981.56   473.7  982.48   483.2  985.93   510.8 1004.51   528.2 1015.01
   549.1 1025.35   557.6 1027.82   569.1 1029.28   639.6 1036.45   661.0 1036.40
   820.6 1021.82   968.9 1031.52  1014.8 1032.18  1090.7 1031.57  1165.9 1028.01
  1307.3 1029.59  1417.6 1035.55  1722.7 1046.52  1870.7 1055.89  1919.8 1063.69
#Mann= 3 , 0 , 0
       0     0.1       0   437.4   0.045       0   452.4     0.1       0
Bank Sta=   437.4,   452.4
Exp/Cntr=0.3,0.1

Type RM Length L Ch R = 1 ,7769.9,684.532,688.199,692.467
XS GIS Cut Line= 3
     1713273.754      252319.760     1713977.815      252241.531
     1714925.256      252119.842
#Sta/Elev= 30
       0 1109.64    41.7 1095.44    93.5 1083.09   192.5 1066.47   417.2 1034.49
   558.0 1023.12   606.6 1017.36   627.2 1012.42   682.8  982.74   693.4  979.67
   703.6  979.23   717.0  978.87   718.6  978.99   830.0  987.65   848.5  991.20
   897.3 1006.55   987.1 1019.42  1012.9 1021.08  1135.0 1014.66  1160.4 1011.15
  1187.9 1002.99  1201.8 1001.37  1223.4 1004.30  1237.3 1008.34  1275.5 1013.18
  1297.2 1013.96  1345.6 1023.05  1470.0 1035.26  1517.4 1038.45  1663.6 1042.40
#Mann= 3 , 0 , 0
       0     0.1       0   703.6   0.045       0   718.6     0.1       0
Bank Sta=   703.6,   718.6
Exp/Cntr=0.3,0.1

Type RM Length L Ch R = 1 ,7081.7,676.743,681.258,680.564
XS GIS Cut Line= 3
     1713265.062      252545.755     1714368.961      252710.906
     1714986.101      252806.519
#Sta/Elev= 30
       0 1103.94   120.7 1074.08   184.5 1060.19   222.7 1053.53   304.1 1045.28
   398.8 1028.86   467.5 1023.77   524.6 1021.09   581.7 1020.78   614.9 1023.00
   784.3 1014.32   855.0 1005.74   927.0  987.48   958.4  981.24  1102.2  975.50
  1107.1  975.38  1117.2  976.64  1131.1  981.76  1141.5  988.82  1179.2 1019.07
  1186.9 1024.40  1199.6 1030.80  1237.1 1035.82  1255.1 1039.58  1281.6 1040.42
  1376.4 1048.14  1472.3 1059.07  1511.9 1066.11  1628.7 1093.19  1740.7 1110.46
#Mann= 3 , 0 , 0
       0     0.1       0  1102.2   0.045       0  1117.2     0.1       0
Bank Sta=  1102.2,  1117.2
Exp/Cntr=0.3,0.1

Type RM Length L Ch R = 1 ,6400.5,302.672,304.589,311.631
XS GIS Cut Line= 3
     1713099.911      252702.214     1713819.011      253033.871
     1714273.347      253188.972
#Sta/Elev= 30
       0 1135.06    66.7 1109.85    88.9 1103.24   282.5 1058.31   341.6 1053.51
   367.3 1052.68   385.2 1048.54   416.7 1039.03   459.7 1028.90   530.7 1018.81
   588.5 1013.58   671.6 1008.95   689.5 1004.53   712.7  993.82   745.3  981.29
   763.2  976.55   784.4  972.99   795.9  972.18   799.4  972.71   890.6  985.57
   910.8  990.33   946.7 1007.65   974.2 1015.76  1012.2 1023.95  1045.3 1027.43
  1055.1 1030.42  1088.5 1035.82  1105.7 1038.28  1179.5 1043.73  1272.0 1042.36
#Mann= 3 , 0 , 0
       0     0.1       0   784.4   0.045       0   799.4     0.1       0
Bank Sta=   784.4,   799.4
Exp/Cntr=0.3,0.1

Type RM Length L Ch R = 1 ,6095.9,514.874,495.411,471.637
XS GIS Cut Line= 3
     1712981.532      252945.492     1713700.632      253277.149
     1713821.936      253311.870
#Sta/Elev= 30
       0 1069.55    67.2 1066.10   117.5 1060.86   154.5 1056.16   184.4 1048.93
   201.6 1047.41   214.3 1047.87   249.7 1045.40   267.4 1045.44   291.1 1043.93
   312.4 1043.84   324.1 1043.13   375.3 1034.17   394.2 1030.20   441.0 1022.75
   501.5 1015.22   576.4 1007.16   628.9  999.05   635.3  995.80   642.0  994.05
   646.2  991.74   652.7  984.77   667.3  971.24   672.7  969.20   675.9  968.97
   682.3  969.17   725.3  978.08   791.9  984.57   851.0  989.62   918.1 1000.04
#Mann= 3 , 0 , 0
       0     0.1       0   667.3   0.045       0   682.3     0.1       0
Bank Sta=   667.3,   682.3
Exp/Cntr=0.3,0.1

Type RM Length L Ch R = 1 ,5600.5,407.054,384.922,367.102
XS GIS Cut Line= 3
     1712952.145      253858.265     1713422.451      253644.702
     1713991.061      253242.683
#Sta/Elev= 30
       0 1146.59    18.6 1141.85    35.1 1139.22    90.0 1135.11   109.8 1130.58
   172.6 1111.80   234.6 1091.75   301.4 1066.65   338.0 1053.91   363.1 1043.35
   437.8 1007.38   471.4  992.11   501.0  974.09     509  970.32   511.3  969.29
   520.1  968.57     524  969.64   550.7  977.57   574.1  980.95   608.1  984.33
   663.6  985.80   715.2  991.53   866.9  993.98   894.6  992.01   925.1  992.55
  1039.4 1004.38  1107.9 1005.78  1155.8 1009.41  1170.3 1012.15  1212.9 1027.42
#Mann= 3 , 0 , 0
       0     0.1       0     509   0.045       0     524     0.1       0
Bank Sta=     509,     524
Exp/Cntr=0.3,0.1

Type RM Length L Ch R = 1 ,5215.5,806.043,815.078,831.794
XS GIS Cut Line= 3
     1713721.999      254088.305     1713837.311      253419.495
     1714014.233      253257.990
#Sta/Elev= 30
       0 1036.41    54.1 1033.86   118.3 1034.87   142.4 1033.14   186.1 1027.70
   263.3 1021.21   275.0 1019.80   302.7 1014.03   347.2 1001.24   354.3  998.09
   359.3  995.12   382.3  972.68   386.8  970.56   395.4  966.81   401.8  967.70
   431.1  971.88   491.8  976.68   528.0  988.62   552.1  991.00   614.1  993.91
   687.0 1000.13   716.6 1001.76   764.2 1001.86   809.0 1003.67   823.7 1004.99
   839.8 1009.21   859.5 1018.76   883.3 1026.34   888.0 1027.47   918.2 1031.68
#Mann= 3 , 0 , 0
       0     0.1       0   386.8   0.045       0   401.8     0.1       0
Bank Sta=   386.8,   401.8
Exp/Cntr=0.3,0.1

Type RM Length L Ch R = 1 ,4400.5,558.979,562.062,557.736
XS GIS Cut Line= 3
     1713830.049      254414.561     1714476.759      253403.534
     1714867.856      253061.625
#Sta/Elev= 30
       0 1038.15    73.4 1033.31   134.1 1031.86   216.8 1026.32   275.2 1025.19
   397.4 1018.92   446.7 1015.61   571.2 1011.50   679.9 1012.07   706.0 1012.89
   795.3 1010.33   828.5 1007.92   861.1 1004.51   959.4  991.14  1059.8  983.25
  1085.6  982.30  1192.7  966.35  1196.4  965.89  1207.7  967.80  1213.3  969.11
  1269.4  992.52  1313.1 1014.86  1329.1 1024.30  1346.2 1032.86  1388.5 1043.54
  1525.2 1072.09  1590.7 1090.26  1633.6 1103.70  1705.0 1120.91  1719.6 1123.63
#Mann= 3 , 0 , 0
       0     0.1       0  1192.7   0.045       0  1207.7     0.1       0
Bank Sta=  1192.7,  1207.7
Exp/Cntr=0.3,0.1

Type RM Length L Ch R = 1 ,3838.4,311.348,317.385,322.687
XS GIS Cut Line= 3
     1714151.658      254605.787     1714864.411      253780.036
     1715199.354      253420.229
#Sta/Elev= 30
       0 1031.39   137.1 1029.34   290.3 1022.87   347.2 1022.57   596.2 1019.93
   666.5 1018.25   759.2 1017.00   784.1 1016.03   807.5 1015.94   868.2 1009.12
   882.1 1006.71   908.5 1001.13   916.1  998.87   945.1  991.91   988.2  980.79
  1001.3  976.51  1013.7  974.23    1068  965.98  1072.9  965.29    1083  966.93
  1085.5  967.40  1101.8  974.47  1166.5  995.47  1177.2 1000.25  1204.4 1014.32
  1237.2 1032.00  1291.3 1057.61  1464.4 1125.77  1552.8 1157.44  1582.4 1168.88
#Mann= 3 , 0 , 0
       0     0.1       0    1068   0.045       0    1083     0.1       0
Bank Sta=    1068,    1083
Exp/Cntr=0.3,0.1

Type RM Length L Ch R = 1 ,3521,315.749,320.553,322.732
XS GIS Cut Line= 3
     1714290.731      254553.634     1715020.869      254058.184
     1715434.032      253761.200
#Sta/Elev= 30
       0 1029.72   143.9 1027.21   239.7 1024.97   385.0 1024.89   420.5 1024.02
   440.1 1024.04   552.2 1016.93   619.0 1015.05   632.8 1013.74   656.6 1009.14
   691.1 1001.80   750.6  985.06   794.1  973.33   807.1  969.38   844.5  964.10
   879.1  960.41   880.3  960.48   895.3  961.48   904.2  962.14   935.9  969.35
   946.6  974.09  1005.8 1005.09  1031.5 1015.42  1077.3 1034.83  1097.7 1042.37
  1140.3 1059.67  1167.4 1073.24  1194.3 1085.20  1347.0 1148.93  1391.2 1169.11
#Mann= 3 , 0 , 0
       0     0.1       0   880.3   0.045       0   895.3     0.1       0
Bank Sta=   880.3,   895.3
Exp/Cntr=0.3,0.1

Type RM Length L Ch R = 1 ,3200.5,413.308,400,387.101
XS GIS Cut Line= 3
     1714368.961      254666.632     1715148.988      254344.607
     1715602.629      254081.673
#Sta/Elev= 30
       0 1028.44    85.3 1023.46   207.6 1020.73   240.1 1016.08   264.9 1014.07
   327.7 1018.34   425.3 1015.47   619.0 1006.83   671.8  997.77   683.9  994.77
   708.1  993.16   725.3  989.36   743.4  982.00   768.8  970.00   793.3  965.44
   836.4  961.23   845.6  960.31   851.4  961.08   878.8  965.24   917.9  969.50
   931.6  973.63   958.2  989.10   988.6  999.73  1043.2 1017.06  1083.6 1028.05
  1137.7 1038.09  1195.7 1052.39  1254.2 1074.32  1347.3 1102.45  1368.2 1110.02
#Mann= 3 , 0 , 0
       0     0.1       0   836.4   0.045       0   851.4     0.1       0
Bank Sta=   836.4,   851.4
Exp/Cntr=0.3,0.1

Type RM Length L Ch R = 1 ,2800.5,688.412,678.673,671.611
XS GIS Cut Line= 3
     1715194.712      254944.780     1715429.658      254611.022
     1715733.623      254075.568
#Sta/Elev= 30
       0 1014.54     3.3 1016.62     5.6 1016.96    50.2 1020.59    63.5 1021.23
    90.3 1018.47   135.2 1009.78   148.9 1005.20   236.1  969.64   257.8  967.06
   373.4  965.64   380.5  965.11   400.7  961.42   406.1  960.39   415.7  961.14
   425.3  963.94   440.8  969.37   474.8  988.74   490.8  993.94   520.3 1000.58
   551.1 1006.15   650.4 1027.12   759.0 1052.60   796.4 1062.50   833.5 1070.56
   855.6 1076.45   889.9 1082.24   959.0 1103.15   982.9 1111.28  1023.9 1126.15
#Mann= 3 , 0 , 0
       0     0.1       0   400.7   0.045       0   415.7     0.1       0
Bank Sta=   400.7,   415.7
Exp/Cntr=0.3,0.1

Type RM Length L Ch R = 1 ,2121.8,220.111,217.691,215.367
XS GIS Cut Line= 3
     1715782.240      255379.799     1715832.293      255157.773
     1715989.801      254295.866
#Sta/Elev= 30
       0 1024.66    60.2 1021.75    77.5 1021.22   104.7 1018.95   210.0 1007.21
   232.0 1001.61   238.5  998.31   271.9  978.75   286.7  971.09   306.1  963.93
   310.9  962.45     324  960.98   331.5  960.09     339  960.84   342.6  961.19
   369.3  967.65   391.4  970.84   425.5  972.11   552.1  974.70   636.8  979.13
   667.0  985.91   673.0  986.81   805.7 1002.85   838.1 1007.29   935.2 1028.85
   991.3 1040.87  1017.0 1045.80  1029.5 1047.48  1071.3 1055.53  1103.8 1062.60
#Mann= 3 , 0 , 0
       0     0.1       0     324   0.045       0     339     0.1       0
Bank Sta=     324,     339
Exp/Cntr=0.3,0.1

Type RM Length L Ch R = 1 ,1904.1,398.141,398.529,399.057
XS GIS Cut Line= 3
     1716028.239      255564.298     1716058.989      255103.050
     1716133.460      254179.873
#Sta/Elev= 30
       0 1027.09    44.7 1028.13    96.4 1022.73   241.4 1011.41   250.6 1011.18
   279.6 1009.10   298.1 1008.86   313.2 1005.51   357.9  986.86   387.0  976.36
   438.8  961.52   441.9  960.64   453.8  960.76   496.5  968.01   531.1  971.68
   583.0  973.24   821.1  974.90   900.6  980.29   954.1  987.24  1008.9 1000.66
  1057.5 1013.44  1074.2 1015.25  1109.0 1020.80  1152.0 1026.53  1167.0 1030.87
  1198.7 1038.71  1252.4 1051.13  1299.5 1059.43  1327.9 1066.43  1388.4 1089.16
#Mann= 3 , 0 , 0
       0     0.1       0   438.8   0.045       0   453.8     0.1       0
Bank Sta=   438.8,   453.8
Exp/Cntr=0.3,0.1

Type RM Length L Ch R = 1 ,1505.6,1131.704,1148.147,1164.354
XS GIS Cut Line= 3
     1716427.987      255464.361     1716455.069      255127.314
     1716385.532      254153.797
#Sta/Elev= 30
       0 1024.90    25.8 1025.04    68.2 1023.34   105.3 1019.78   151.6 1013.01
   184.6 1005.07   219.3  991.42   272.8  971.27   289.3  963.21   293.6  961.70
   306.4  960.45   308.6  960.78   325.7  963.38   335.6  964.18   457.0  970.57
   478.7  970.94   542.7  969.73   810.8  967.92   878.4  970.85   896.3  973.50
   965.3  992.37  1063.3 1022.29  1086.1 1026.72  1104.7 1032.57  1122.8 1034.33
  1150.0 1040.35  1178.2 1045.84  1215.1 1056.66  1292.5 1076.34  1314.1 1085.82
#Mann= 3 , 0 , 0
       0     0.1       0   293.6   0.045       0   308.6     0.1       0
Bank Sta=   293.6,   308.6
Exp/Cntr=0.3,0.1

Type RM Length L Ch R = 1 ,357.4,354.707,356.96,356.568
XS GIS Cut Line= 4
     1716497.174      255479.736     1716843.110      255233.737
     1717245.884      254851.533     1717525.859      254465.709
#Sta/Elev= 30
       0 1022.79    36.7 1023.36    57.1 1022.38   101.6 1021.41   230.9 1020.60
   285.4 1019.41   506.1 1013.28   665.9 1006.30   755.3 1000.42   761.7 1000.41
   786.9  999.06   811.1  995.77   824.8  992.43   906.6  969.78   929.6  957.80
   932.5  957.44   945.8  955.78   947.5  956.16   970.6  962.88  1013.5  973.90
  1053.9  989.61  1073.7  998.74  1128.6 1022.67  1180.4 1047.17  1221.0 1068.15
  1284.7 1102.46  1317.5 1118.98  1388.1 1151.35  1405.8 1159.10  1456.4 1178.91
#Mann= 3 , 0 , 0
       0     0.1       0   932.5   0.045       0   947.5     0.1       0
Bank Sta=   932.5,   947.5
Exp/Cntr=0.3,0.1

Type RM Length L Ch R = 1 ,0.5,0,0.457,7.325
XS GIS Cut Line= 4
     1716541.990      255622.765     1717154.956      255373.982
     1717401.929      255183.222     1717828.423      254770.937
#Sta/Elev= 30
       0 1015.34   113.9 1015.46   181.7 1017.51   417.8 1015.18   659.6 1002.32
   690.6 1001.39   776.0  996.28   802.9  993.12   836.9  985.97   863.3  982.42
   922.8  972.52   943.3  967.20   963.7  957.38   966.1  956.73   972.1  955.36
   981.1  956.42   988.1  957.36  1041.8  971.91  1085.6  987.00  1117.2  997.22
  1135.1 1004.16  1160.9 1012.94  1183.8 1018.24  1230.6 1027.07  1257.6 1034.41
  1335.3 1064.65  1370.7 1080.92  1450.1 1114.98  1522.2 1144.21  1566.8 1159.38
#Mann= 3 , 0 , 0
       0     0.1       0   966.1   0.045       0   981.1     0.1       0
Bank Sta=   966.1,   981.1
Exp/Cntr=0.3,0.1
